--- 67_ras.prj (project) ---

Proj Title=67
Current Plan=p01
Default Exp/Contr=0.3,0.1
English Units
Geom File=g01
Flow File=f01
Plan File=p01
Y Axis Title=Elevation
X Axis Title(PF)=Main Channel Distance
X Axis Title(XS)=Station
BEGIN DESCRIPTION:
RFD model 67 exported to HEC-RAS
END DESCRIPTION:

--- 67_ras.p01 (plan) ---

Plan Title=Plan 01
Program Version=4.10
Short Identifier=Plan 01
Geom File=g01
Flow File=f01
Subcritical Flow
Calc Critical at every XS
Secant Critical Depth

--- 67_ras.f01 (steady flow) ---

Flow Title=Flow 01
Program Version=5.01
Number of Profiles= 6
Profile Names=10yr,25yr,50yr,100yr,100plus,500yr
River Rch & RM=67,50,14130.59
   89.33  168.89  254.11  347.52  507.39 1147.15
River Rch & RM=67,50,13897.32
   92.93  175.73  264.46  361.73  528.12 1187.58
River Rch & RM=67,50,13664.05
   97.77  184.94  278.37   380.8  555.97 1241.43
River Rch & RM=67,50,13340.05
  116.73  221.08  333.09  455.92  665.65  1450.6
River Rch & RM=67,50,13186.26
  122.68  232.43  350.29  479.56  700.16 1515.54
River Rch & RM=67,50,12810.85
  126.21  239.17  360.52  493.62  720.69 1553.99
River Rch & RM=67,50,12589.39
  128.95  244.41  368.45  504.52   736.6 1583.63
River Rch & RM=67,50,12367.93
  129.92  246.26  371.27  508.39  742.25 1594.16
River Rch & RM=67,50,12146.47
  133.79  253.65  382.49  523.82  764.78 1636.03
River Rch & RM=67,50,12067.85
  135.71  257.33  388.07   531.5  775.99  1656.8
River Rch & RM=67,50,11915.39
  136.29  258.43  389.74   533.8  779.35 1663.02
River Rch & RM=67,50,11593.88
  151.24  287.05   433.2  593.61  866.66 1823.52
River Rch & RM=67,50,11345.77
  153.43  291.27  439.64   602.5  879.64  1847.4
River Rch & RM=67,50,11097.67
  155.06  294.42  444.44  609.13  889.33 1865.24
River Rch & RM=67,50,10849.56
  280.11   533.2  806.65 1106.73 1615.82 3120.03
River Rch & RM=67,50,10601.45
  281.86  536.59  811.83 1113.91  1626.3 3137.79
River Rch & RM=67,50,10346.19
  284.55  541.81  819.82 1124.98 1642.47 3165.16
River Rch & RM=67,50,10169.45
  285.19  543.04   821.7 1127.58 1646.27 3171.58
River Rch & RM=67,50,9958.208
  287.24  547.02   827.8 1136.03  1658.6 3192.43
River Rch & RM=67,50,9746.962
  306.88  584.97  885.82 1216.26 1775.75 3388.71
River Rch & RM=67,50,9535.716
  307.66  586.48  888.13 1219.47 1780.42 3396.53
River Rch & RM=67,50,9324.469
  307.82  586.78  888.59 1220.11 1781.36  3398.1
River Rch & RM=67,50,9142.982
   312.6  596.07  902.83 1239.85 1810.18 3446.42
River Rch & RM=67,50,8961.168
  314.11  599.01  907.36 1246.15 1819.38 3461.94
River Rch & RM=67,50, 8804.17
  314.41  599.59  908.26 1247.41 1821.21 3465.05
River Rch & RM=67,50,8517.069
  329.82   629.7  954.62 1311.92  1915.4  3623.4
River Rch & RM=67,50,8361.211
  330.55  631.14  956.84 1315.02 1919.93 3631.02
River Rch & RM=67,50,8180.868
  331.73  633.45   960.4 1319.98 1927.16 3643.19
River Rch & RM=67,50,8037.211
  349.99  668.92 1014.82 1395.47 2037.39 3825.44
River Rch & RM=67,50,7832.822
  350.56  670.05 1016.57 1397.91 2040.94  3831.4
River Rch & RM=67,50,7628.432
  352.99  674.82 1023.96 1408.24 2056.03 3856.72
River Rch & RM=67,50,7424.043
   354.7  678.19 1029.17 1415.52 2066.67 3874.55
River Rch & RM=67,50,7061.587
  356.12  680.99 1033.51 1421.59 2075.52 3889.38
River Rch & RM=67,50,6771.846
  371.83   711.7 1080.82 1487.45 2171.68  4048.2
River Rch & RM=67,50,6571.956
  372.97  713.94 1084.27 1492.27 2178.72 4059.87
River Rch & RM=67,50,6396.007
  373.97  715.89 1087.29 1496.49 2184.88 4070.07
River Rch & RM=67,50,6133.012
   374.8  717.54 1089.84 1500.07  2190.1  4078.8
River Rch & RM=67,50,5996.464
  377.15  722.19 1097.06 1510.19 2204.87  4103.5
River Rch & RM=67,50,5797.199
  377.98  723.83 1099.61 1513.76 2210.08 4112.21
River Rch & RM=67,50,5556.358
  378.39  724.64 1100.88 1515.53 2212.68 4116.56
River Rch & RM=67,50,5216.189
  385.38   738.5 1122.41 1545.74 2256.77 4190.23
River Rch & RM=67,50,5064.175
  385.79  739.31 1123.67 1547.51 2259.36 4194.54
River Rch & RM=67,50,4913.114
  387.83  743.36 1129.97 1556.35 2272.27 4216.11
River Rch & RM=67,50,4764.347
   388.1   743.9 1130.81 1557.53 2273.99 4218.98
Boundary for River Rch & Prof#=67,50,1
Up Type= 0
Dn Type= 2
Boundary for River Rch & Prof#=67,50,2
Up Type= 0
Dn Type= 2
Boundary for River Rch & Prof#=67,50,2
Up Type= 0
Dn Type= 2
Boundary for River Rch & Prof#=67,50,2
Up Type= 0
Dn Type= 2
Boundary for River Rch & Prof#=67,50,2
Up Type= 0
Dn Type= 2
Boundary for River Rch & Prof#=67,50,2
Up Type= 0
Dn Type= 2

--- 67_ras.g01 (geometry) ---

Geom Title=67
Program Version=4.10

River Reach=67,50
Reach XY= 30
989261.311374815762713.490028123989090.255676735761320.439482827
989481.248898479761016.972030669989597.973508392760596.860953462
989151.186868817760174.166378174989691.128976005759828.173196287
989704.822090254 759694.80938926 990004.14934297759642.233842987
990007.084591049759479.049637775990168.760872679759501.905514416
990280.902139249759304.301757479990490.436911553759380.411688268
990572.963199348759194.498436888 990357.61678787758956.073163373
990786.673548358758250.848745055990430.157714267758173.216920389
990479.144565643757919.831843914990303.363315615757574.779760575
990474.009772081 757568.30532407990420.082413915757103.329389552
990586.853706989757061.069576531990824.939675452756747.128678372
990822.665831194756505.264286719 991374.11119658756034.158613083
991122.219548837755718.095898051 991324.37309793755095.472816136
991228.432255644754733.582334729991433.706034199754439.042887209
991460.362294931753055.555890377991825.855608747752413.915311435

Type RM Length L Ch R = 1 ,14130.59,233.273500,233.273500,233.273500
XS GIS Cut Line= 6
989394.358141937762746.257114555989308.471746296  762729.1477464
989243.183650129762705.320697906989218.386228836762698.744979995
989176.402883734762693.926819016989127.011186033762693.115443789
#Sta/Elev= 29
9862.745304.15719872.243301.23379882.394298.64749892.544295.95939912.845 289.377
9923.099 285.7419943.648279.25989950.356276.99469953.998 275.655 9964.49 270.985
9974.981267.81019978.207267.0542 9985.67265.12939993.569262.52349996.445261.7018
    9999261.7292   10001261.842510007.22262.713910021.15266.948410038.71273.6185
10045.55276.076110048.96 277.03310069.09 280.347 10078.4281.445610089.22282.0496
10099.22282.485610109.22283.190110129.22285.074110137.21 286.153
#Mann= 3 , 0 , 0
9862.745    0.12       09862.745    0.12       010137.21    0.12       0
#XS Ineff= 2 , 0
       0                               0
Bank Sta=9862.745,10137.21
Exp/Cntr=0.3,0.1

Type RM Length L Ch R = 1 ,13897.32,233.273500,233.273500,233.273500
XS GIS Cut Line= 6
989392.342239473762502.039265905 989295.92676442762503.006034003
989216.969170051762490.609913328 989191.56222055762488.544465585
989157.311252289762489.117864005989109.866188707 762493.76217692
#Sta/Elev= 28
9858.076 287.3239865.421286.68079885.429284.63649905.438282.72229915.442281.3488
9925.446279.85749935.449278.07969945.451275.7734 9955.46272.61489965.522266.4878
9975.584259.96859985.708254.16119995.854248.8846   10001250.3885   10006252.1601
10009.71252.886710016.17253.907410026.33 256.10510036.46259.069710046.49261.1077
10056.53263.424210076.54 268.40910086.54270.3149 10106.6272.357910116.65272.3291
 10126.7271.184910136.75 271.182 10141.9271.7236
#Mann= 3 , 0 , 0
9858.076    0.12       09858.076    0.12       0 10141.9    0.12       0
#XS Ineff= 2 , 0
       0                               0
Bank Sta=9858.076,10141.9
Exp/Cntr=0.3,0.1

Type RM Length L Ch R = 1 ,13664.05,324.000000,324.000000,324.000000
XS GIS Cut Line= 6
 989338.44418188 762250.20228705989278.248656071762253.256576758
989232.567591957762260.807216689989202.267448415762270.107253665
989120.478545041762300.837667268989052.573195406762320.070328281
#Sta/Elev= 27
9851.912260.81669865.373260.74369875.386260.84239895.412261.24839905.425261.2117
9915.477261.50749925.613261.66249935.749261.71399945.884261.4419 9956.02260.2546
9958.486259.29299966.402255.61229976.862 249.2869987.322246.49039997.944242.5358
10003.99243.192810019.32246.2838   10030247.924410040.68248.835510051.36250.6414
10072.72257.891110083.25261.799610093.64264.629510104.03 265.81510114.43267.1098
10124.82268.141510148.13269.9335
#Mann= 3 , 0 , 0
9851.912    0.12       09851.912    0.12       010148.13    0.12       0
#XS Ineff= 2 , 0
       0                               0
Bank Sta=9851.912,10148.13
Exp/Cntr=0.3,0.1

Type RM Length L Ch R = 1 ,13340.05,153.789800,153.789800,153.789800
XS GIS Cut Line= 6
989406.425440982 761979.24149279989246.954549041761978.907459203
989235.252351846761979.231950495989202.846203998761980.813444801
989147.021245743761988.841834109989064.644291711762006.780681816
#Sta/Elev= 30
9827.822250.92769839.248248.89059849.248 247.4539859.248246.90879869.248247.0308
9879.248247.37159899.248246.73759909.248 246.2739919.248  247.039929.248 247.435
9949.248247.64649959.248246.84329969.248244.56699979.248239.25899989.249234.4886
9999.253234.744610009.27236.862410029.29243.180410039.37245.887710049.47248.1948
10059.58249.402710069.68250.297510087.84250.707110100.15250.672310110.38251.0003
10130.85251.208310141.08 251.54410151.32251.594510161.55 251.31310172.15 251.565
#Mann= 3 , 0 , 0
9827.822   0.055       09827.822   0.055       010172.15   0.055       0
#XS Ineff= 2 , 0
       0                               0
Bank Sta=9827.822,10172.15
Exp/Cntr=0.3,0.1

Type RM Length L Ch R = 1 ,13186.26,153.789800,153.789800,153.789800
XS GIS Cut Line= 6
989373.192018393761798.260138635989305.230985532761809.516331825
989177.757927855761837.613337564989156.021986778761851.067405584
989099.932927218761900.988839971989050.112818043761932.277369428
#Sta/Elev= 30
 9820.41 239.5339828.713239.2777 9838.85238.64149848.986237.48049859.122235.6904
9869.258238.25219879.394239.79889889.533240.61829899.751240.84039909.969241.2365
9920.188240.96499930.406241.80249950.843242.2517 9971.28 242.0669981.498238.4267
9991.716233.010910001.91231.369510012.32231.813810022.97233.115610035.21233.7022
10045.54234.820810065.97237.679610074.27239.300410080.64240.858410090.13242.8147
10101.05244.414210111.29245.400710150.87246.763110162.39246.708910179.54246.9288
#Mann= 3 , 0 , 0
 9820.41    0.12       0 9820.41    0.12       010179.54    0.12       0
#XS Ineff= 2 , 0
       0                               0
Bank Sta=9820.41,10179.54
Exp/Cntr=0.3,0.1

Type RM Length L Ch R = 1 ,13032.47,221.613500,221.613500,221.613500
XS GIS Cut Line= 2
989206.774868846761726.950288296988976.306118816761854.554454952
#Sta/Elev= 28
9865.794237.47579879.254237.78249882.413237.61769890.684237.00929903.058236.4624
9913.545235.56569924.975234.28599936.406233.39139947.836232.99739959.267232.3306
9964.992231.84469970.697230.85959982.128229.65069993.558228.817510004.99226.9629
10006.28226.927510016.42228.176310027.85234.363510039.28 239.63610047.57240.0557
10050.71240.117210062.14239.988210068.22240.522510073.57240.8984   10085 241.372
10109.51242.729810119.29243.192610129.23243.3446
#Mann= 3 , 0 , 0
9865.794  0.1084       09865.794  0.1084       010129.23  0.1084       0
#XS Ineff= 2 , 0
       0                               0
Bank Sta=9865.794,10129.23
Exp/Cntr=0.3,0.1

Type RM Length L Ch R = 1 ,12810.85,221.461000,221.461000,221.461000
XS GIS Cut Line= 2
989187.243618846761582.419038281988955.472785473761634.502371654
#Sta/Elev= 30
9892.419228.78589894.718228.72469904.191229.03739904.968229.06719915.217228.6747
9925.467228.68049935.716228.10739945.965 227.622  9949.8227.37299956.215226.7718
9966.464225.86049976.713225.22719986.963222.5893 9995.41221.31679997.212221.0304
10007.46220.213110017.71225.450410027.96228.743610038.21230.856210041.02230.9057
10048.46230.947910058.71230.831310068.96230.432710079.21230.237610086.63230.0607
10089.46229.984510099.71230.441910109.96230.8548 10120.2231.229710129.97232.1358
#Mann= 3 , 0 , 0
9892.419    0.12       09892.419    0.12       010129.97    0.12       0
#XS Ineff= 2 , 0
       0                               0
Bank Sta=9892.419,10129.97
Exp/Cntr=0.3,0.1

Type RM Length L Ch R = 1 ,12589.39,221.461100,221.461100,221.461100
XS GIS Cut Line= 6
989297.823741548761445.453175724 989210.82563952761410.675579063
989159.418779217761396.542212994989109.743725013761390.302393771
989015.307428829761390.397477649988932.843735493761380.626906647
#Sta/Elev= 30
 9812.64 220.2869815.681219.91919826.451217.5378 9837.22215.54119847.989217.4001
9858.759220.04639869.528221.55949880.298221.84519891.067221.54039901.836221.4149
9912.445220.93419922.939219.94359933.432219.37349943.732218.54739953.979217.6094
9964.154 216.4769974.239214.41259984.324211.59469994.409208.390310004.55208.7449
10014.56210.243610024.57212.566310044.57217.581810064.58221.351810074.59224.0487
 10084.6224.618810104.61226.970510144.89230.691110154.96231.840210187.34233.4367
#Mann= 3 , 0 , 0
 9812.64    0.12       0 9812.64    0.12       010187.34    0.12       0
#XS Ineff= 2 , 0
       0                               0
Bank Sta=9812.64,10187.34
Exp/Cntr=0.3,0.1

Type RM Length L Ch R = 1 ,12367.93,221.461000,221.461000,221.461000
XS GIS Cut Line= 6
989322.308359114761386.181662865989287.995778924 761360.71771421
989255.916710878761330.358741156989145.175940467761179.095021246
989112.881529338761144.781546108989070.700614703761109.055915829
#Sta/Elev= 30
9811.513218.50549854.242210.17079872.134207.45399885.903212.45159891.656212.9103
9917.935212.67679932.282213.17389950.602212.89779954.595212.57999966.409210.1236
9978.222206.35829988.017203.68179990.319202.6671    9999199.727810003.46199.0449
10016.55203.787310019.07 204.46910029.05207.8454 10035.9210.339310041.48212.7301
10052.74217.121410066.34219.195710105.47 223.592 10119.2224.639710130.14224.9883
10143.56225.235210148.36225.031110156.66224.305610169.77223.708810188.51221.7443
#Mann= 3 , 0 , 0
9811.513    0.12       09811.513    0.12       010188.51    0.12       0
#XS Ineff= 2 , 0
       0                               0
Bank Sta=9811.513,10188.51
Exp/Cntr=0.3,0.1

Type RM Length L Ch R = 1 ,12146.47,78.618000,78.618000,78.618000
XS GIS Cut Line= 2
989324.830424368761157.071816087989320.924174368761035.978066072
#Sta/Elev= 14
9942.965200.02299945.038199.68889955.044198.86119965.049197.34849975.054196.0139
9985.059194.83349995.064193.859710005.07193.557710015.07194.586610025.08196.4608
10035.09197.574610045.09198.8531 10055.1201.629210064.12203.2789
#Mann= 3 , 0 , 0
9942.965    0.12       09942.965    0.12       010064.12    0.12       0
#XS Ineff= 2 , 0
       0                               0
Bank Sta=9942.965,10064.12
Exp/Cntr=0.3,0.1

Type RM Length L Ch R = 1 ,12067.85,152.463800,152.463800,152.463800
XS GIS Cut Line= 2
989422.920702169761138.408621624989368.233202139761001.689871624
#Sta/Elev= 21
9926.343203.61579930.015203.46469940.785202.56139947.671201.58989951.555200.9534
9962.326 198.5119973.096194.83219974.596194.17679983.866189.15089994.637186.6405
10001.52187.112510005.41187.500310016.18 191.00410026.95194.219110028.45194.5099
10037.72196.397910048.49198.406310055.37199.700810059.26200.276210070.03200.7835
10073.59200.9951
#Mann= 3 , 0 , 0
9926.343    0.04       09926.343    0.04       010073.59    0.04       0
#XS Ineff= 2 , 0
       0                               0
Bank Sta=9926.343,10073.59
Exp/Cntr=0.3,0.1

Type RM Length L Ch R = 1 ,11915.39,73.408400,73.408400,73.408400
XS GIS Cut Line= 2
989598.701952159760984.762788281989424.222785473760961.325288281
#Sta/Elev= 22
9903.055199.0176 9906.79198.6751 9916.88197.0959 9926.97196.3189 9937.06 195.461
 9947.15194.15869957.239191.88019967.329 188.4899976.386186.22579977.419185.9768
9987.509183.31899997.599 182.82910007.69182.453310017.78185.354610027.87188.4261
10037.96189.825710048.05 192.021 10051.5192.805810058.14194.297310068.23196.3591
10078.32197.6386 10079.1197.7182
#Mann= 3 , 0 , 0
9903.055    0.04       09903.055    0.04       0 10079.1    0.04       0
#XS Ineff= 2 , 0
       0                               0
Bank Sta=9903.055,10079.1
Exp/Cntr=0.3,0.1

Type RM Length L Ch R = 1 ,11841.98,248.105400,248.105400,248.105400
XS GIS Cut Line= 2
989586.983202189760909.241954952989441.149868846760889.710704967
#Sta/Elev= 19
9922.508192.58029924.508192.52519934.598192.19279944.687191.38819954.464190.2638
9954.776190.22789964.866187.89269974.955184.30089985.044178.94559995.133174.3877
10005.22175.566210015.31 181.327 10025.4186.2055 10029.8 187.72510035.49189.6441
10045.58192.048210055.67 193.89910065.76194.824910069.64194.9861
#Mann= 3 , 0 , 0
9922.508    0.04       09922.508    0.04       010069.64    0.04       0
#XS Ineff= 2 , 0
       0                               0
Bank Sta=9922.508,10069.64
Exp/Cntr=0.3,0.1

Type RM Length L Ch R = 1 ,11593.88,248.105500,248.105500,248.105500
XS GIS Cut Line= 6
989797.877183696760713.497753394989667.678918332760685.888868311
989558.451720117760656.918796462989517.788687132760649.583327016
989449.806304327760649.573388427989377.312731397760662.860813162
#Sta/Elev= 30
9785.348182.10379788.289181.89589798.511182.55119808.734183.53539829.178184.9786
9849.623185.57059870.068185.3872 9880.29185.03589890.513184.53629910.957182.7511
9921.211182.15589952.225177.08079962.563174.10929972.901171.5456 9983.24 166.671
9993.578160.375310000.69160.064210003.93160.2701 10014.3162.818610024.66163.5122
10065.44 173.33610075.56176.158910085.57178.236710095.59180.826110105.61182.2704
10125.63183.528210165.89 183.21910176.06183.438510186.29 183.99910214.59184.5283
#Mann= 3 , 0 , 0
9785.348    0.04       09785.348    0.04       010214.59    0.04       0
#XS Ineff= 2 , 0
       0                               0
Bank Sta=9785.348,10214.59
Exp/Cntr=0.3,0.1

Type RM Length L Ch R = 1 ,11345.77,248.105400,248.105400,248.105400
XS GIS Cut Line= 6
989695.998634823760341.139124598989622.645326316760373.764776021
989488.787471023760462.498864502989462.156039073760487.006119197
989401.077955234760558.435516328 989353.82064755760600.537943825
#Sta/Elev= 30
 9782.71165.73399794.451165.70229838.062166.15429849.268166.69419872.094168.2134
9884.528169.46899895.597170.35769907.663169.75049931.795 169.9329938.807168.8604
9943.861167.45129955.928162.73679967.994159.2267 9980.06154.56019992.126151.3244
    9999150.731510004.19150.569910016.24153.077810027.43154.595810042.47155.4041
10056.96157.049110070.94159.9696 10083.6163.665210096.76 168.41510123.07174.2373
10132.49175.563310136.23175.943710147.87176.631110202.81178.330410217.25179.2043
#Mann= 3 , 0 , 0
 9782.71    0.04       0 9782.71    0.04       010217.25    0.04       0
#XS Ineff= 2 , 0
       0                               0
Bank Sta=9782.71,10217.25
Exp/Cntr=0.3,0.1

Type RM Length L Ch R = 1 ,11097.67,248.105500,248.105500,248.105500
XS GIS Cut Line= 6
989418.806835499760205.064508642989377.620683849  760231.3458709
989350.435779467760263.370415977989314.029286363760332.408923957
989267.190624608760461.898040568989181.318980425760559.934639809
#Sta/Elev= 30
9780.763162.89939785.125 162.6089796.586159.09289808.046 154.9469820.304152.3823
9829.774152.54689848.046155.07319861.277  161.279873.743164.60719885.314163.7617
9896.884164.55369930.732 165.0549941.789  162.419952.733  157.429963.356 151.177
9973.979147.89739984.352147.06759994.661143.7451   10005142.9077 10015.4 147.131
10025.81 153.87310036.32158.041110047.16157.840410092.26167.152710103.65168.9242
   10111169.853710153.58172.860410167.38173.113310188.03174.497710219.27175.7955
#Mann= 3 , 0 , 0
9780.763    0.04       09780.763    0.04       010219.27    0.04       0
#XS Ineff= 2 , 0
       09921.032                       0
Bank Sta=9780.763,10219.27
Exp/Cntr=0.3,0.1

Type RM Length L Ch R = 1 ,10849.56,248.105400,248.105400,248.105400
XS GIS Cut Line= 6
989503.749678876760179.975384685989443.604015293760187.771864969
989331.565835384760206.880663415989120.723805662 760226.66182216
988962.292195352760226.297789229988784.249933371760213.857862777
#Sta/Elev= 30
9638.467164.7744 9647.29162.38839667.457159.64759687.624158.89549697.708161.6468
9707.868163.15669718.041162.71719728.214159.60439738.387153.92199758.733145.4224
9779.039143.27539799.233143.16329829.414141.65539919.764 144.5389970.072144.5973
10010.28135.870410040.32 137.24810070.33141.464510110.33144.254610120.33143.6067
10130.34141.123710140.34140.023110150.34143.201210160.34147.728510200.37169.5897
10210.39172.696110240.43178.059710270.48181.565410300.57184.946210361.55190.1012
#Mann= 3 , 0 , 0
9638.467    0.12       09638.467    0.12       010361.55    0.12       0
#XS Ineff= 2 , 0
       09949.316        10031.34       0
Bank Sta=9638.467,10361.55
Exp/Cntr=0.3,0.1

Type RM Length L Ch R = 1 ,10601.45,255.267800,255.267800,255.267800
XS GIS Cut Line= 6
989625.475009691760181.538225831989469.145672642760161.185583503
 989408.89318007760137.725060789 989354.78989125 760096.50799542
989148.084813525759909.253845975989021.863291358759815.402911962
#Sta/Elev= 30
 9636.57159.67559707.549161.56539727.692162.96489757.942162.90589768.066161.0217
9778.189161.70199788.313158.87799798.575157.50629852.297152.64819900.821150.0215
9913.997151.14669926.932149.31859944.599148.01879959.712145.49519974.825140.5914
9989.938131.77299993.611130.5119   10001130.024910005.08130.096610026.14 134.284
10034.98137.476110049.56147.398910061.32154.043410064.13155.155510078.71 157.941
10122.43158.719610167.15160.933910273.87161.745410298.52 164.63310363.51164.0329
#Mann= 3 , 0 , 0
 9636.57    0.12       0 9636.57    0.12       010363.51    0.12       0
#XS Ineff= 2 , 0
       09944.461                       0
Bank Sta=9636.57,10363.51
Exp/Cntr=0.3,0.1

Type RM Length L Ch R = 1 ,10346.19,176.732200,176.732200,176.732200
XS GIS Cut Line= 4
989495.886244535 760012.20970659989495.886244535759927.258159101
989535.634216309759846.982843608989477.181316704759757.355064154
#Sta/Elev= 26
9890.992153.41779898.201151.50669908.201147.12539918.201 142.5429928.201138.3152
9938.201135.48329948.201132.40479958.201 130.3879968.201129.90269989.622129.5085
10000.78129.3164 10023.1129.246610045.42129.327310066.68129.554910067.89129.6112
10079.83131.134110091.76134.2689 10103.7137.544210115.64141.6925 10121.6144.5358
10127.58147.130210139.91150.887910151.46155.839310158.21158.2799 10163.4158.8717
10172.52158.8345
#Mann= 3 , 0 , 0
9890.992  0.1128       09890.992  0.1128       010172.52  0.1128       0
#XS Ineff= 2 , 0
       0                               0
Bank Sta=9890.992,10172.52
Exp/Cntr=0.3,0.1

Type RM Length L Ch R = 1 ,10169.45,211.246200,211.246200,211.246200
XS GIS Cut Line= 6
989906.465456301760120.559310169989845.323332654760065.741036423
989784.809253912759999.084417047989652.650235844759815.509431765
989543.545166889759727.451970629989403.970479869759590.603362909
#Sta/Elev= 30
9632.797151.14029783.981148.55449835.333 145.9989885.761146.94919936.411146.2512
9948.134144.97649954.048142.72529971.685130.71099984.009120.78449991.303117.7539
9995.629117.298910007.25119.121210019.29123.236410027.66124.338610041.61 134.745
10080.05134.0282 10096.8132.338110129.41136.183710143.46137.070610169.81155.8198
10175.23157.6146 10203.8157.349910218.08154.579410232.36154.307210239.71155.0817
10253.72159.933310260.93160.041510275.22156.9963 10289.5155.0089 10367.2146.0286
#Mann= 3 , 0 , 0
9632.797  0.0636       09632.797  0.0636       0 10367.2  0.0636       0
#XS Ineff= 2 , 0
       0                               0
Bank Sta=9632.797,10367.2
Exp/Cntr=0.3,0.1

Type RM Length L Ch R = 1 ,9958.208,211.246200,211.246200,211.246200
XS GIS Cut Line= 6
989953.612977511759982.685517243989759.887178524759728.879278494
989730.673712637759631.751021349989689.733817063759560.327437132
 989620.36054827759476.407527602989531.336964474759386.953467122
#Sta/Elev= 30
9630.578142.21199652.464143.84079677.214143.55249713.102142.45869763.839138.7865
9800.965140.83499838.602140.86189890.989139.77629904.086137.96589930.113128.4349
9941.354124.93179954.295121.13369976.045115.68719996.498109.39899998.579109.3903
10006.69109.8965 10016.9124.907210027.35 134.84710037.89138.074110081.65142.6596
10093.15143.2459 10116.9 143.21710128.77145.937310134.32146.567610166.39146.5458
10286.85135.024910336.57131.460610350.47129.325910364.38126.217810369.48125.5353
#Mann= 3 , 0 , 0
9630.578    0.12       09630.578    0.12       010369.48    0.12       0
#XS Ineff= 2 , 0
       0                               0
Bank Sta=9630.578,10369.48
Exp/Cntr=0.3,0.1

Type RM Length L Ch R = 1 ,9746.962,211.246200,211.246200,211.246200
XS GIS Cut Line= 6
990085.478069887759992.254975328990002.433313749759872.689649705
989956.457716085759777.030282676989938.113320993  759696.7169182
989945.870546995759592.825846797989707.402723116759349.073919772
#Sta/Elev= 30
9608.909151.13879655.406 146.7319712.551  139.379751.847130.98669774.665129.8014
9797.367126.4983 9819.54127.23789841.287134.9703 9852.16136.51549873.364137.5063
9894.207136.80249904.629133.18059924.924121.09229935.032116.62329945.123 113.835
9955.132111.717210006.18106.385410016.48 107.96910026.71115.506610081.22117.8673
10121.87121.396510132.37123.699110149.26131.588610163.29134.242410217.38137.0231
10244.97137.048410263.92138.632410272.56140.753210313.94137.699710391.09129.7774
#Mann= 3 , 0 , 0
9608.909    0.12       09608.909    0.12       010391.09    0.12       0
#XS Ineff= 2 , 0
       0                               0
Bank Sta=9608.909,10391.09
Exp/Cntr=0.3,0.1

Type RM Length L Ch R = 1 ,9535.716,211.246200,211.246200,211.246200
XS GIS Cut Line= 6
990249.551631944759792.439542395990134.036040307759633.751169604
990042.042900329759527.021290584989953.126259039759484.458588716
 989909.44018402 759454.58934756989697.668915438759249.721944903
#Sta/Elev= 30
9607.885128.12349617.087123.90479632.611 124.5689649.602120.94199666.562119.1045
9678.931119.5624  9691.3116.99739700.577113.02239716.038116.14389728.407121.5951
 9734.56121.73639740.776121.10039777.882111.42389802.527109.08739854.254110.0564
9894.031107.43519966.618106.19839998.693101.649810009.44 102.08210020.25110.6462
 10031.3124.439810042.35131.979210053.95132.888110130.34133.010510170.19 134.355
10186.09137.004810226.51136.209910313.27126.950510382.04123.525210392.12122.0259
#Mann= 3 , 0 , 0
9607.885    0.12       09607.885    0.12       010392.12    0.12       0
#XS Ineff= 2 , 0
       09851.631                       0
Bank Sta=9607.885,10392.12
Exp/Cntr=0.3,0.1

Type RM Length L Ch R = 1 ,9324.469,181.487700,181.487700,181.487700
XS GIS Cut Line= 4
990330.472785503759596.741954952990214.587368876759518.616954952
990030.993618816759426.169038281989932.035285503759348.044038281
#Sta/Elev= 30
9814.825134.77159845.545131.63559857.606129.70129869.666125.89149881.726120.4346
9893.786117.02319917.907114.79239925.277114.63399943.166111.95879954.087111.1154
9965.319109.55119976.516105.92429987.712 101.3519998.908 97.6462 10007.197.10902
 10010.197.42273 10021.3102.519210029.33104.7127 10032.5105.163310043.69104.9574
10066.09106.677410088.48110.682310099.67113.201410144.46127.992710155.66129.9315
10167.78130.399710210.44130.405710231.48131.168510258.86130.065110286.22130.2718
#Mann= 3 , 0 , 0
9814.825    0.12       09814.825    0.12       010286.22    0.12       0
#XS Ineff= 2 , 0
       0                               0
Bank Sta=9814.825,10286.22
Exp/Cntr=0.3,0.1

Type RM Length L Ch R = 1 ,9142.982,181.813200,181.813200,181.813200
XS GIS Cut Line= 2
990358.671909988759522.035845101990153.810798854759174.813622862
#Sta/Elev= 30
9782.777126.22289802.556 123.4039814.167120.38179825.778116.63349837.389112.3018
 9849.04108.7857 9860.61106.1181 9868.72104.61679888.399103.10079908.078102.0968
9930.275101.84699947.437102.13689965.107100.43339976.71899.607199988.32997.01244
 9999.9495.3963210006.4796.6051810011.5598.2769810023.1699.9511710034.77  102.15
10045.83104.669610057.99108.105210065.51109.1894 10069.6109.431310085.19111.3251
10092.83112.537310127.66120.180210150.88121.9143 10174.1121.369310185.93121.5406
#Mann= 3 , 0 , 0
9782.777    0.12       09782.777    0.12       010185.93    0.12       0
#XS Ineff= 2 , 0
       0                               0
Bank Sta=9782.777,10185.93
Exp/Cntr=0.3,0.1

Type RM Length L Ch R = 1 ,8961.168,156.998600,156.998600,156.998600
XS GIS Cut Line= 2
990374.296909988 759492.52195619990384.713576645759308.494178399
#Sta/Elev= 21
9884.088123.73889891.622123.06359896.529122.34749901.638121.61769911.654119.8482
 9921.67117.92879931.686115.27619941.702 111.6959951.718106.69149961.734101.7346
 9971.7599.809049981.766 99.93099991.78296.65808 10001.894.0041910011.81 93.8488
10021.8396.4127210031.8599.9527410041.86105.290710051.88109.714310061.89  113.62
10068.41115.3543
#Mann= 3 , 0 , 0
9884.088    0.12       09884.088    0.12       010068.41    0.12       0
#XS Ineff= 2 , 0
       0                               0
Bank Sta=9884.088,10068.41
Exp/Cntr=0.3,0.1

Type RM Length L Ch R = 1 , 8804.17,287.101000,287.101000,287.101000
XS GIS Cut Line= 3
990731.514452159759441.794038281990631.233129829759397.566941783
990379.505243272759277.244178399
#Sta/Elev= 30
9755.178129.06749773.227128.52459795.086127.60289806.015127.40749860.662124.9783
9871.688124.76529916.022122.48149927.106121.0982 9938.19117.76499949.273111.9683
9960.357105.94659971.441101.38639982.52498.119829986.67295.911429993.60892.66246
10004.6991.8682110009.8693.7450910015.78 96.549610026.8699.7724710033.0599.84619
10049.0399.0181610071.1999.9445710079.42101.604610082.28102.422210104.44  111.09
10115.53114.5042 10125.8 117.13310126.61117.2664 10137.7117.353110143.79116.7578
#Mann= 3 , 0 , 0
9755.178    0.12       09755.178    0.12       010143.79    0.12       0
#XS Ineff= 2 , 0
       0                               0
Bank Sta=9755.178,10143.79
Exp/Cntr=0.3,0.1

Type RM Length L Ch R = 1 ,8517.069,155.858000,155.858000,155.858000
XS GIS Cut Line= 3
990584.379035532759056.377371624990508.131775498759079.335030153
990400.338576645 759242.52195619
#Sta/Elev= 30
9852.368113.02299862.163113.27159872.607113.26139893.494113.82369903.937 114.005
 9914.38 113.9129924.824113.61789931.997112.97399937.679112.05219938.786111.8006
9950.771106.67429955.822103.69469962.75599.981469973.96695.243379986.72591.33616
9992.109 89.94199998.70988.5954910010.2592.7006510022.6897.92691 10028.499.88616
10034.66101.193710046.54103.868510064.68106.408710070.62107.0251 10082.6108.5637
10094.59109.498410100.97110.404810106.57111.032910119.11112.762310127.57113.2548
#Mann= 3 , 0 , 0
9852.368  0.0743       09852.368  0.0743       010127.57  0.0743       0
#XS Ineff= 2 , 0
       0                               0
Bank Sta=9852.368,10127.57
Exp/Cntr=0.3,0.1

Type RM Length L Ch R = 1 ,8361.211,180.342500,180.342500,180.342500
XS GIS Cut Line= 6
990775.068446837758944.149233066990582.501562488758952.965197205
990374.206178518759018.996922813 990256.01507032759040.846748209
990129.673757525759016.995084358989969.765028505758949.816874095
#Sta/Elev= 30
9582.295109.44429602.383108.86659622.403106.84639642.419102.26259662.422104.9192
9682.425105.64599732.642102.4984  9793.5101.21779813.974101.66839855.422104.6163
9897.381106.56599927.805106.68159940.033105.08589950.751100.0832 9961.4796.27868
9993.62587.6292410003.91  88.98210024.5496.7097910055.48109.857510065.78113.1442
10075.89114.567410106.04115.156410136.07116.807510156.21116.8036 10176.5113.1107
10196.97114.647210207.29116.6962 10238.6117.541210346.17118.131110417.68117.1769
#Mann= 3 , 0 , 0
9582.295    0.06       09582.295    0.06       010417.68    0.06       0
#XS Ineff= 2 , 0
       0                               0
Bank Sta=9582.295,10417.68
Exp/Cntr=0.3,0.1

Type RM Length L Ch R = 1 ,8180.868,143.657500,143.657500,143.657500
XS GIS Cut Line= 5
990759.405059308 758854.65958856990657.135774165758842.682104722
990494.979069829758855.580933481990374.282886416758849.131519094
990236.081149757758859.266313136
#Sta/Elev= 30
9638.993107.09679643.429106.42949653.497104.40489663.565 102.1559673.634100.3816
9683.70299.21407 9693.7798.824319703.83999.268929722.03599.140269804.29496.59606
9824.35796.340749834.38996.425699874.51595.377319884.54695.389029914.62494.84125
9934.652 94.80019964.695 95.03119994.73895.7258310014.7796.3908110034.8197.54527
10054.8698.3826310074.9198.0697210084.94 98.424110094.97 99.909910104.99 102.862
10115.02 105.52810125.05108.602110135.08109.852210155.13110.692710164.07111.3242
#Mann= 3 , 0 , 0
9638.993    0.12       09638.993    0.12       010164.07    0.12       0
#XS Ineff= 2 , 0
       0                               0
Bank Sta=9638.993,10164.07
Exp/Cntr=0.3,0.1

Type RM Length L Ch R = 1 ,8037.211,204.389400,204.389400,204.389400
XS GIS Cut Line= 6
990834.438620824758858.822474375990706.653708736758826.080673364
990630.557693195758801.242754621990458.810113435758721.998215212
990235.691519703758639.462068492 990005.02365542758577.578747118
#Sta/Elev= 30
9560.998107.43369591.388107.9705 9632.68106.95169673.972100.8782 9705.1799.88769
9726.20897.974469736.72897.768569747.24798.175259789.798104.4359 9822.27106.5315
9886.653107.40519899.712108.81879910.829107.72269944.182107.35039955.299104.9573
9966.218100.87959976.816 93.71459987.41383.891259998.01180.1291210019.0682.15039
10050.9188.9096310072.3395.2639210093.75103.9127 10100.9105.831910147.31110.5937
10184.66113.009210263.59112.8362 10346.4 110.65310377.29110.434810439.04107.8985
#Mann= 3 , 0 , 0
9560.998    0.06       09560.998    0.06       010439.04    0.06       0
#XS Ineff= 2 , 0
       0                               0
Bank Sta=9560.998,10439.04
Exp/Cntr=0.3,0.1

Type RM Length L Ch R = 1 ,7832.822,204.389400,204.389400,204.389400
XS GIS Cut Line= 6
990953.360534743758776.005331563990750.673092924758694.624493697
990486.699705571758518.487437259990421.347207434758484.650333467
990323.040156822758462.123810365990155.207923164758449.185854738
#Sta/Elev= 30
9560.325104.08219600.686104.31539632.413105.43689655.876 104.9419675.118102.4048
9683.359102.12019707.671103.21359740.804101.79039763.097103.06699778.217101.9904
9797.366102.22539809.042 103.5569820.718103.75969855.768103.2293 9868.05 103.938
9929.457103.83429941.739 99.58219959.12487.808289978.39178.1740610002.2778.47557
10014.3177.4679910026.3583.3498510038.3993.2007810048.9596.4414910074.51100.7878
10121.57100.716110166.2698.6948810208.3297.9090110369.7297.6286510439.6796.31051
#Mann= 3 , 0 , 0
9560.325    0.12       09560.325    0.12       010439.67    0.12       0
#XS Ineff= 2 , 0
       0                               0
Bank Sta=9560.325,10439.67
Exp/Cntr=0.3,0.1

Type RM Length L Ch R = 1 ,7628.432,204.389400,204.389400,204.389400
XS GIS Cut Line= 6
 991080.31166046758621.451500849990932.953760586758572.785582934
990827.241101114 758521.74585594 990629.20758667758359.797258707
990416.897959857758408.976585099990282.676614438758422.433003133
#Sta/Elev= 30
9557.63199.140329584.06798.870149636.288100.09929721.56499.556989732.48297.14717
 9787.6698.722929798.965100.48319810.26998.622969821.57497.736129868.45496.87436
9922.39897.729999944.07596.889579966.31685.938689973.30283.317099987.06375.40114
10000.7971.6512110014.6676.2020110028.5484.6691410057.5987.9761310070.1788.75621
10081.4489.1742210105.9788.52472 10143.189.6812710174.5191.3864810226.8796.59432
10237.3496.8897410288.7195.7930410309.1696.34292 10369.794.6174110442.2295.19172
#Mann= 3 , 0 , 0
9557.631    0.12       09557.631    0.12       010442.22    0.12       0
#XS Ineff= 2 , 0
       0                               0
Bank Sta=9557.631,10442.22
Exp/Cntr=0.3,0.1

Type RM Length L Ch R = 1 ,7424.043,362.455300,362.455300,362.455300
XS GIS Cut Line= 2
 990952.24015826758133.171140924990619.174589813758351.177694783
#Sta/Elev= 30
9799.63987.933249844.14788.512619856.09986.883239868.05187.231019880.00286.85077
9891.95487.163559894.27686.861579903.906 85.05569915.85782.498849927.80981.07505
9939.76180.395719949.05579.637659963.66478.061339975.616 74.96849985.57471.17485
9987.56870.638149999.51968.9477310011.4772.4614210022.09 74.014910023.4274.16377
10040.3574.2528510047.33 74.703510076.8779.3450810095.13 82.447510130.9982.93692
10149.9183.8310810166.8485.3180210178.7986.1144810190.7587.2429310197.7187.65365
#Mann= 3 , 0 , 0
9799.639    0.12       09799.639    0.12       010197.71    0.12       0
#XS Ineff= 2 , 0
       0                               0
Bank Sta=9799.639,10197.71
Exp/Cntr=0.3,0.1

Type RM Length L Ch R = 1 ,7061.587,289.741000,289.741000,289.741000
XS GIS Cut Line= 2
990594.783021063 758088.00806728990370.824687749758288.528900638
#Sta/Elev= 28
9821.18788.685079831.66988.489859847.74187.531789874.58682.596869888.009 81.2651
9901.43180.755389928.27680.574169936.60980.259159941.69979.80612  9951.678.65326
9955.12278.406819966.59276.585629981.58370.342989996.57566.6488110008.8165.35096
10011.5766.3010210022.2374.1602310026.5677.8830210035.6683.6601310041.5585.61767
10049.0887.2761810056.5488.53967 10062.589.2818410075.92 90.459510089.3591.32548
10101.5191.1967110116.1991.29271 10121.891.46052
#Mann= 3 , 0 , 0
9821.187  0.0605       09821.187  0.0605       0 10121.8  0.0605       0
#XS Ineff= 2 , 0
       0                               0
Bank Sta=9821.187,10121.8
Exp/Cntr=0.3,0.1

Type RM Length L Ch R = 1 ,6771.846,199.890500,199.890500,199.890500
XS GIS Cut Line= 2
990607.803854376 757931.75806728990269.262187719 758002.07056728
#Sta/Elev= 30
9861.20284.668029864.066 84.81499874.27984.427049894.70682.88368 9904.9281.64075
9915.13379.410319925.34777.91118 9935.5677.457759945.77376.206779955.98773.32928
  9966.269.747369976.41466.880019986.627 65.6226 9996.8463.3380810007.0563.45266
10017.2764.1533410037.69 70.520610047.9172.4504810058.1273.5574310068.3374.02775
10078.5574.9485410088.7676.6816510098.9778.9496210123.0282.8378310129.6183.37101
10139.8383.5614710160.2583.1933710170.47 83.414110201.1185.5776610206.9786.36241
#Mann= 3 , 0 , 0
9861.202    0.12       09861.202    0.12       010206.97    0.12       0
#XS Ineff= 2 , 0
       0                               0
Bank Sta=9861.202,10206.97
Exp/Cntr=0.3,0.1

Type RM Length L Ch R = 1 ,6571.956,175.948800,175.948800,175.948800
XS GIS Cut Line= 2
990511.449687749757788.528900623990206.762187719757877.070567295
#Sta/Elev= 30
 9844.0380.471989861.16180.250939881.98881.029399892.40280.440779902.81580.57037
9913.22980.316979923.64379.049219934.05676.85567 9938.8976.11728 9944.4775.43577
9954.884 75.07489965.29770.391899974.72666.563899975.71166.251129986.125 62.1394
9996.53860.1919710006.9563.7621810017.3772.9432310027.7879.0662610038.1980.34629
10048.6181.2274110059.0281.2709110069.4381.5177210082.2381.3720710090.2681.61613
10100.6882.61307 10121.582.6868710142.3383.81091 10153.984.7885910161.3285.31596
#Mann= 3 , 0 , 0
 9844.03   0.055       0 9844.03   0.055       010161.32   0.055       0
#XS Ineff= 2 , 0
       0                               0
Bank Sta=9844.03,10161.32
Exp/Cntr=0.3,0.1

Type RM Length L Ch R = 1 ,6396.007,262.995300,262.995300,262.995300
XS GIS Cut Line= 2
990479.765659958757650.942095071990212.838576645757674.813622862
#Sta/Elev= 26
9831.33476.367389836.11976.398689846.15976.064419866.23975.551959876.27972.77511
9886.31871.779559896.35871.382049906.39871.372229916.43871.874429936.51871.78606
9946.55870.206229956.59867.475079966.63865.360249976.67864.231129986.71861.78017
9996.75858.08644 10006.858.8492210016.8463.5150110026.8865.3803110046.9671.06369
   1005774.6381210067.0477.4193710077.0878.7569710087.1279.1760110097.1679.25139
10099.3379.17935
#Mann= 3 , 0 , 0
9831.334  0.0758       09831.334  0.0758       010099.33  0.0758       0
#XS Ineff= 2 , 0
       0                               0
Bank Sta=9831.334,10099.33
Exp/Cntr=0.3,0.1

Type RM Length L Ch R = 1 ,6133.012,136.548000,136.548000,136.548000
XS GIS Cut Line= 4
990525.338576645757644.431678414 990390.78996554757525.074039519
990301.814271092757507.712928399990236.710104406757518.563622847
#Sta/Elev= 30
 9908.86 75.92149923.07275.806879949.41574.93715 9953.2174.905759962.78375.63421
9968.27975.485439976.15173.532119983.348 69.51619989.51862.720549998.41754.76212
10002.8954.7049710013.4958.0499810016.2558.8512610029.6261.7676610042.9966.76802
10058.6969.0076410069.7269.9774910073.7670.2064110083.0970.9084610088.7270.98762
10094.62 70.6454   1011571.1842210125.1871.8646310135.3771.9136610155.7572.51254
10179.3772.5312910206.5673.0390610226.8372.5405810236.9773.0218110245.3872.90952
#Mann= 3 , 0 , 0
 9908.86    0.12       0 9908.86    0.12       010245.38    0.12       0
#XS Ineff= 2 , 0
       0                               0
Bank Sta=9908.86,10245.38
Exp/Cntr=0.3,0.1

Type RM Length L Ch R = 1 ,5996.464,199.264900,199.264900,199.264900
XS GIS Cut Line= 2
990629.505243301757459.969872862990241.050382197757462.140011728
#Sta/Elev= 30
9827.14671.094579841.65171.035129851.65270.668849871.65271.016459881.65270.75668
9901.65270.639559921.65369.775589941.65368.547669951.653 67.03699961.65365.96783
9971.65364.517959981.65461.149339991.65456.9286310001.6553.2524110011.6554.99366
10021.6558.7604410031.6562.1715410041.6563.4973810051.6563.2602410061.6564.29315
10071.6664.4773110081.6665.3118910091.6665.9014710101.6666.2469210111.6666.35363
10131.6667.0335510141.6667.1223610151.6667.6730410181.6668.4029610215.6169.56731
#Mann= 3 , 0 , 0
9827.146  0.0727       09827.146  0.0727       010215.61  0.0727       0
#XS Ineff= 2 , 0
       0                               0
Bank Sta=9827.146,10215.61
Exp/Cntr=0.3,0.1

Type RM Length L Ch R = 1 ,5797.199,240.841300,240.841300,240.841300
XS GIS Cut Line= 2
990591.923770607757282.340007052990307.304103017757258.117056608
#Sta/Elev= 28
9857.18466.890739864.13266.847549874.16967.125869884.20567.044319904.27767.59282
9914.31367.378499924.34967.953029934.385 68.30759944.42268.230539954.45868.34591
9964.49467.73397 9974.5359.445729984.56653.014629994.60251.6456610004.6451.43083
10014.6755.0073310024.71  62.61710034.7566.3915310044.7867.6574810054.8268.02639
10064.8668.1023810084.9367.2221310094.9666.92897   1010566.8353110115.04 67.3919
10125.0767.0536110135.1167.0389310142.8367.75595
#Mann= 3 , 0 , 0
9857.184    0.12       09857.184    0.12       010142.83    0.12       0
#XS Ineff= 2 , 0
       0                               0
Bank Sta=9857.184,10142.83
Exp/Cntr=0.3,0.1

Type RM Length L Ch R = 1 ,5556.358,340.169000,340.169000,340.169000
XS GIS Cut Line= 2
 990547.03996554757171.341400638990388.619826615756965.178206176
#Sta/Elev= 29
9849.73464.779429853.08264.835479857.73164.781919870.34365.298999882.95464.35228
9885.90664.340869902.31863.699969908.17763.75007 9918.7362.780349920.78862.52778
  9933.4 59.57039946.01156.961519958.62255.144989967.96654.403499971.23454.22938
9983.84552.530419984.379 52.39569996.45747.7332310000.7947.2940610009.0748.25271
 10017.253.8690910021.6856.8561510033.6163.4946110034.2963.7411910059.5164.68227
10082.8564.9645410084.74 64.893210097.3564.8553510109.7364.28832
#Mann= 3 , 0 , 0
9849.734    0.12       09849.734    0.12       010109.73    0.12       0
#XS Ineff= 2 , 0
       0                               0
Bank Sta=9849.734,10109.73
Exp/Cntr=0.3,0.1

Type RM Length L Ch R = 1 ,5216.189,152.013700,152.013700,152.013700
XS GIS Cut Line= 2
 990898.60246554757021.601817295990477.595521092756769.865706176
#Sta/Elev= 30
9781.08360.582679796.93160.453769808.583 58.83519820.23459.191149831.88558.73331
9843.53760.665829855.18861.197189866.83959.670259901.79359.779189936.747 59.0014
 9960.0559.416729971.701 59.30149983.35254.269849995.00442.9462310006.6543.01465
10018.3148.3526810027.7852.1378210041.6158.3020510053.2659.2591110064.9159.38945
10076.5659.8474510088.2159.7869310099.8760.0494810123.1759.8157910169.77 60.4122
10181.4259.9958810222.6361.1087610251.3360.5928510262.9861.2467410271.6161.17871
#Mann= 3 , 0 , 0
9781.083    0.12       09781.083    0.12       010271.61    0.12       0
#XS Ineff= 2 , 0
       0                               0
Bank Sta=9781.083,10271.61
Exp/Cntr=0.3,0.1

Type RM Length L Ch R = 1 ,5064.175,151.060400,151.060400,151.060400
XS GIS Cut Line= 2
990902.858115554756850.326630726990633.642970711756684.354187042
#Sta/Elev= 30
 9871.2558.729839880.48157.471479892.22956.919659903.97756.035279927.47255.94093
9938.56655.996019950.96756.539829957.62156.515769962.71556.383599974.463 53.7532
 9986.2146.763949995.73241.881929997.958 41.195310009.7142.4838110021.45 54.8912
10033.8456.8957210044.9557.58419 10052.957.5778810071.9557.2160510080.1956.95707
10091.9457.1932210110.0656.6793310115.4356.6722310129.1257.3222210138.9357.50574
10148.1757.4276610167.2357.5793110174.1757.7579610185.9257.3901310187.5257.47371
#Mann= 3 , 0 , 0
 9871.25    0.12       0 9871.25    0.12       010187.52    0.12       0
#XS Ineff= 2 , 0
       0                               0
Bank Sta=9871.25,10187.52
Exp/Cntr=0.3,0.1

Type RM Length L Ch R = 1 ,4913.114,148.767700,148.767700,148.767700
XS GIS Cut Line= 2
990906.778724462756646.454967618990632.336101055756643.841228366
#Sta/Elev= 26
9925.52256.86647  9927.3 56.85499937.30153.424329947.30152.503249957.30252.75042
9977.30353.441969987.303 48.95899997.30439.40698 10007.341.20193 10017.346.45252
 10027.353.5569710037.3155.5306410057.3155.2220410067.3155.3199110077.3155.29027
10087.3155.8991610097.3156.3753510107.3155.8264410127.3156.2543810137.3156.34836
10147.31 56.965310157.3156.5565310167.3156.8361310177.3156.7202310187.3157.30521
10199.9857.63326
#Mann= 3 , 0 , 0
9925.522    0.12       09925.522    0.12       010199.98    0.12       0
#XS Ineff= 2 , 0
       0                               0
Bank Sta=9925.522,10199.98
Exp/Cntr=0.3,0.1

Type RM Length L Ch R = 1 ,4764.347,97.042300,97.042300,97.042300
XS GIS Cut Line= 3
990898.937506616756565.429050252990786.546718031756460.879479423
990585.288794219756319.737558842
#Sta/Elev= 30
9902.67454.008039932.66852.465639949.025 52.10529962.03252.31085 9976.3446.06749
9989.99837.7990810006.0836.0460110020.7636.2817710035.4439.9816610044.6343.52749
10050.12 44.347810058.0643.6331610066.41 39.809910070.2837.5807210082.49 37.7914
10094.71 41.847810118.66 42.925110143.5641.4808710155.7839.4728610167.9938.97561
10170.9139.80797 10180.246.4411810188.3351.2434610192.4251.9045410205.7452.13228
10240.5854.3837410257.9955.1340610277.9255.1953710290.1354.7374910301.9955.20454
#Mann= 3 , 0 , 0
9902.674    0.12       09902.674    0.12       010301.99    0.12       0
#XS Ineff= 2 , 0
       0                 10050.9       0
Bank Sta=9902.674,10301.99
Exp/Cntr=0.3,0.1

Type RM Length L Ch R = 1 ,4667.305,276.710900,276.710900,276.710900
XS GIS Cut Line= 2
990934.282966703757190.922340155990902.131524444756097.773301706
#Sta/Elev= 30
9262.23864.393699358.20262.324139378.21163.131139418.22860.937629498.26260.11371
9508.26758.815549568.29357.155079638.32356.905959728.36254.612659788.38855.07846
9798.39257.148969868.42253.94873 9908.4453.313979928.44854.60849 9978.4735.67323
9988.47433.144519998.47932.3666910018.49 35.454610028.4940.75442 10038.543.15725
10078.5146.6632110098.52 47.441210108.5346.3109310198.5746.4728910218.5750.31529
10228.5848.71977 10278.647.73164 10288.648.9489910318.62 49.116110355.8652.85137
#Mann= 3 , 0 , 0
9262.238    0.12       09262.238    0.12       010355.86    0.12       0
#XS Ineff= 2 , 0
       0                               0
Bank Sta=9262.238,10355.86
Exp/Cntr=0.3,0.1

Type RM Length L Ch R = 1 ,4390.594,493.988900,493.988900,493.988900
XS GIS Cut Line= 2
991571.953239113 756767.59501645990912.848671824756060.263285682
#Sta/Elev= 30
9381.68954.73604 9439.9153.249719523.90652.817269549.25851.826569641.25651.77274
9672.27550.660179685.94451.477969740.61849.881379773.27450.518739795.29248.41619
 9808.9648.057849846.61750.740679863.63449.750699890.97151.540179905.29250.47457
9934.62951.071999945.64648.393189959.31439.503199978.63537.787129993.30431.47395
10000.3229.7168910027.6638.9866710037.3139.8307910068.6640.5693610082.3341.76096
10191.6842.6883110246.3541.8355410260.02 42.490510286.6847.1853510348.5151.23054
#Mann= 3 , 0 , 0
9381.689    0.12       09381.689    0.12       010348.51    0.12       0
#XS Ineff= 2 , 0
       0                               0
Bank Sta=9381.689,10348.51
Exp/Cntr=0.3,0.1

Type RM Length L Ch R = 1 ,3896.605,493.988900,493.988900,493.988900
XS GIS Cut Line= 6
991719.700532389755816.105555871991480.955724874755835.834419109
991395.922904755755874.541578765991219.337769289756004.831165912
991103.414736498756029.147974875990976.321032023756026.921373721
#Sta/Elev= 30
9599.18541.702459633.90541.316859744.06942.28001 9764.2442.722379784.41143.85836
9825.393 43.12949846.18944.106999934.26544.086239950.83131.76392 9959.7528.42934
 9997.8929.0104610040.6428.1729110050.0329.9236510071.0432.2906110107.3834.29743
10126.9136.6470910137.7935.9207810159.3335.5678610169.7333.6304710180.1332.85553
10211.1833.9727910261.7733.8639710301.9334.4576510311.9435.6143910331.9641.13049
10341.9743.1055310351.97 42.723210361.9843.2809610372.0246.7107810400.8347.66675
#Mann= 3 , 0 , 0
9599.185    0.12       09599.185    0.12       010400.83    0.12       0
#XS Ineff= 2 , 0
       0                               0
Bank Sta=9599.185,10400.83
Exp/Cntr=0.3,0.1

Type RM Length L Ch R = 1 ,3402.616,0.000000,0.000000,0.000000
XS GIS Cut Line= 6
991609.283558865 755635.43756942991411.149615823755634.341313153
991315.998948721755618.586770163991261.424073845  755592.7477102
 991107.65744764755488.554053762990864.001048157755397.391300597
#Sta/Elev= 30
9599.10539.632439613.38839.349199663.38840.117969683.38840.755069693.38840.34123
9773.39842.364099843.624 42.01199863.97636.642889874.20935.91335  9884.636.83356
9895.03336.425989916.62331.369979967.49428.1840210001.0124.52824 10012.424.69807
   1002527.16381 10033.929.56405 10037.630.9075210050.3438.8755710062.7942.81177
10109.78 42.478610132.3442.8052510185.6742.7608510226.57 41.882210241.1442.09304
10251.7841.7338610336.4143.1369310368.1442.4798710378.7242.7740310400.9442.11837
#Mann= 3 , 0 , 0
9599.105    0.12       09599.105    0.12       010400.94    0.12       0
#XS Ineff= 2 , 0
       0                               0
Bank Sta=9599.105,10400.94
Exp/Cntr=0.3,0.1
